HEC-RAS study Q100-00-00.prj: Q100-00-00

--- Q100-00-00.g01 (geometry) --- (continued)

Type RM Length L Ch R = 3 ,92216.8 ,,,
BEGIN DESCRIPTION:
Interstate 10
END DESCRIPTION:
Bridge Culvert--1,0,-1,-1, 0
Deck Dist Width WeirC Skew NumUp NumDn MinLoCord MaxHiCord MaxSubmerge Is_Ogee
67.24,268.43,2.6,0, 31, 31, , , .95, 0, 0,0,,
   -3043   -2030   -1332    -205    -113     118     192    1200  2818.4  3909.4
    4606    4636    4834    4860    5016    5170    5196    5226  5354.6  6267.7
  6391.7  6461.3  6620.9  6770.9  6926.9  7046.9  7446.9    8022    9207   11946
   13227
    33.5    31.6    32.3    49.2    29.4    31.7    48.9    31.8    31.8    27.4
      23   25.72   25.72   25.72   26.54   27.07   27.07   24.34    32.9    55.7
    57.2    32.2      27      28    55.4    54.9    46.8      34    29.5   31.64
   30.13
       0       0       0       0       0       0       0       0       0       0
       0       0       0   18.45   19.85   19.88       0       0       0       0
       0       0       0       0       0       0       0       0       0       0
       0
   -3043   -2030   -1332    -205    -113     118     192    1200  2818.4  3909.4
    4606    4636    4834    4860    5016    5170    5196    5226  5354.6  6267.7
  6391.7  6461.3  6620.9  6770.9  6926.9  7046.9  7446.9    8022    9207   11946
   13227
    33.5    31.6    32.3    49.2    29.4    31.7    48.9    31.8    31.8    27.4
      23   25.72   25.72   25.72   26.54   27.07   27.07   24.34    32.9    55.7
    57.2    32.2      27      28    55.4    54.9    46.8      34    29.5   31.64
   30.13
       0       0       0       0       0       0       0       0       0       0
       0       0       0   18.45   19.85   19.88       0       0       0       0
       0       0       0       0       0       0       0       0       0       0
       0
Pier Skew, UpSta & Num, DnSta & Num=  ,4915, 2 ,4915, 2 , 0 , 0 , 0 ,,
    1.78    1.78
       0      21
    1.78    1.78
       0      21
Pier Skew, UpSta & Num, DnSta & Num=  ,4970, 2 ,4970, 2 , 0 , 0 , 0 ,,
    1.78    1.78
       0      21
    1.78    1.78
       0      21
Pier Skew, UpSta & Num, DnSta & Num=  ,5060, 2 ,5060, 2 , 0 , 0 , 0 ,,
    1.78    1.78
       0      21
    1.78    1.78
       0      21
Pier Skew, UpSta & Num, DnSta & Num=  ,5115, 2 ,5115, 2 , 0 , 0 , 0 ,,
    1.78    1.78
       0      21
    1.78    1.78
       0      21
BR Coef=-1 , 1 , 1 ,.9, 0 ,,,.8,0,1.2,0,
WSPro=,,,, 1 ,,,, 0 ,,,, 0 ,,,,-1 ,-1 ,-1 , 0 , 0 , 0 , 0 , 0
BC Design=,, 0 ,, 0 ,,,,,,
BC HTab HWMax=28.48

Type RM Length L Ch R = 1 ,92026.57,201.66,201.94,202.96
XS GIS Cut Line= 6
     3268860.782    13868612.441     3265563.792      13868610.8
     3264926.167      13868610.8     3262958.006    13868613.843
     3262085.871    13868462.522     3257591.868    13866010.315
#Sta/Elev= 30
 1296.78   27.41 1496.06   26.64 1522.09   23.27 1554.26   26.42  1680.7   27.45
 1809.52   25.42 1910.91   28.06 2204.73   26.08 2482.21   27.56 2963.82   26.01
 3797.35    23.7 4035.49    22.7  4624.5    20.3  4709.5    19.2  4879.5    11.7
  4950.5      12  4959.5     8.1  4974.5     6.1  4980.5    -3.4  5008.5    -4.7
  5036.5      -4  5038.5    -1.3  5041.5     8.5  5049.5    10.8  5159.5    18.4
  5229.5    19.7 6081.61   26.64  8591.1   24.7412370.71   27.6513204.23   26.94
#Mann= 7 ,-1 , 0
 1296.78    .068       0 2963.82    .118       0 3797.35    .068       0
 4035.49    .118       0  4950.5     .04       0  5049.5    .118       0
12370.71    .068       0
#XS Ineff= 2 , 0
       0 4787.21   22.82  5200.7       0   24.07
Permanent Ineff=
       F       F
#Block Obstruct= 2 , 0
         1615.38    26.3
Bank Sta=4950.5,5049.5
XS Rating Curve= 0
Exp/Cntr=.5,.3

Type RM Length L Ch R = 1 ,91824.63,333.65,215.22,80.56
XS GIS Cut Line= 6
     3268860.881    13868412.441     3265563.781      13868410.8
     3264926.128      13868410.8     3262906.729    13868413.922
     3262208.994    13868288.097     3257735.512    13865866.671
#Sta/Elev= 30
1304.645   27.82  1479.7   27.76 1579.84   23.16 1743.74   26.71 1800.18   21.97
 1878.77   27.263067.13525.50004 3241.47   24.89 3335.72   18.99 3425.33   21.06
  3535.5   16.133772.12522.729914124.62522.09003  4613.6   20.89    4716    18.6
    4800     9.5  4970.5       9  4994.5     6.1  5000.5    -3.4  5028.5    -4.7
  5056.5      -4    5064     3.9    5096     8.9  5179.5    16.4    5264      19
  6522.4   25.01 6618.84   28.44 6792.94   25.0512349.58   27.3713054.58   25.12
#Mann= 7 ,-1 , 0
1304.645    .068       03067.135    .118       03772.125    .068       0
4124.625    .118       0  4970.5     .04       0    5096    .118       0
12349.58    .068       0
#XS Ineff= 2 ,-1
 6673.6611226.11   27.23 3144.51 3829.82   23.05
Permanent Ineff=
       F       F
#Block Obstruct= 2 , 0
         1892.77   26.6312185.82            27.5
Bank Sta=4970.5,5096
XS Rating Curve= 0
Exp/Cntr=.3,.1

Type RM Length L Ch R = 1 ,91609.41,403.41,846.71,629.47
XS GIS Cut Line= 6
     3269108.122    13867865.758     3265082.632    13868126.181
      3265064.22    13868334.847     3262906.812    13868325.634
     3262430.733     13868161.17     3257912.306    13865780.773
#Sta/Elev= 30
 867.955   27.713150.185   25.563750.77523.560023991.00522.43001 4288.07   20.22
 4400.81   12.41  4522.3    8.99 4573.46    4.01 4686.69   14.81 4753.48   16.96
 4855.93    7.91    4957     8.2    4964     5.3    4973    -3.8    5001    -4.9
    5034      .7    5043     9.2 5206.16   11.07 5286.91   18.02 5537.15   17.25
 5745.02   22.91 6354.29   24.79 6430.25   27.62 6565.43   24.23 6752.09   24.69
 6796.53   27.44 6852.98   24.7411215.35   28.1412519.36   26.8412879.71   26.03
#Mann= 7 ,-1 , 0
 867.955    .068       03150.185    .118       03750.775    .068       0
3991.005    .118       0    4957     .04       0    5043    .118       0
12519.36    .068       0
#XS Ineff= 2 ,-1
 6461.23 7761.99   26.26 4150.29 4754.02   16.86
Permanent Ineff=
       F       F
Bank Sta=4957,5043
XS Rating Curve= 0
Exp/Cntr=.3,.1

Type RM Length L Ch R = 1 ,90762.7 ,378.79,637.38,541.97
XS GIS Cut Line= 3
     3269095.845    13867589.875     3262811.596    13867754.339
      3258076.77    13865538.406
#Sta/Elev= 30
  739.78   27.38 1509.37   26.69  1567.3    28.6 1623.57   26.73 3272.88   24.61
 3618.31   22.93 3963.73      22 4697.22   21.24 4771.66   18.76 4846.86    9.36
    4957     8.2    4964     5.3    4973    -3.8    5001    -4.9    5024    -2.6
    5034      .7    5037     4.3    5068     3.2 5173.51   12.34    5788   12.44
 5987.27   22.64 6245.07   26.66  6542.8   22.31 6577.07   24.67 6688.76   24.37
 6722.32   27.13 6781.61   24.15  8327.1   27.13 12023.6   27.5612253.89      27
#Mann= 7 ,-1 , 0
  739.78    .068       0 3272.88    .118       0 3618.31    .068       0
 3963.73    .118       0    4957     .04       0    5037    .118       0
 12023.6    .068       0
#XS Ineff= 1 ,-1
 6281.17 7770.17   25.87
Permanent Ineff=
       F
Bank Sta=4957,5037
XS Rating Curve= 0
Exp/Cntr=.3,.1

Type RM Length L Ch R = 1 ,90125.32,518.8,798.84,497.33
XS GIS Cut Line= 5
     3268967.352    13867213.098     3265140.969    13867315.476
     3265114.326    13867218.302     3265091.752    13867090.277
     3263071.921    13867324.675
#Sta/Elev= 30
1006.765   27.51 1727.87   26.92 1789.05   29.03  1845.7   26.993565.36523.48001
3687.20523.15001 3990.19   19.36 4087.52   12.674113.63514.15969 4276.08   21.16
 4670.67   20.27 4824.26    8.99    4935    10.1    4976     3.6    4985    -3.8
    5010    -9.7    5040    -4.8    5050     7.1    5065    10.9 5168.87   10.49
 5243.11   16.01 5293.29   14.93 5348.58    8.59 5825.74   19.57 6250.11   23.31
 6360.32   19.56 6406.33      23 6793.68   22.96 6997.13   27.94 7098.67   25.63
#Mann= 6 ,-1 , 0
1006.765    .068       03565.365    .118       03687.205    .068       0
4113.635    .118       0    4935     .04       0    5065    .118       0
#XS Ineff= 1 ,-1
 3721.27 4286.06   21.06
Permanent Ineff=
       F
#Block Obstruct= 2 , 0
                         7007.33           27.39
Bank Sta=4935,5065
XS Rating Curve= 0
Exp/Cntr=.3,.1

Type RM Length L Ch R = 1 ,89326.48,482.88,658.59,78.03
XS GIS Cut Line= 4
     3266957.988    13866776.877     3265456.798    13866786.469
     3265154.642    13866517.886     3263040.906    13866936.988
#Sta/Elev= 30
3249.975   25.85 3973.25    24.4 4399.15   20.914427.48519.56066 4549.07    8.34
 4665.29    6.77 4723.52    9.48 4861.67   10.52    4951     8.1    4960       7
    4970    -7.5    5000    -9.2    5024    -4.7    5038     5.5    5061     4.3
 5119.23   14.94 5151.56   19.18 5263.37   21.06  5387.2   20.03 5546.58   21.15
 5637.32   19.43  5827.6   18.92 6418.08   20.11 6471.65    18.3 6580.08   20.55
  6660.3   20.07 6714.54   15.43 6738.12   19.83 6767.62   22.53 7310.36    24.9
#Mann= 4 ,-1 , 0
3249.975    .068       04427.485    .118       0    4951     .04       0
    5038    .118       0
#XS Ineff= 1 ,-1
 6585.02 6841.78   20.02
Permanent Ineff=
       F
Bank Sta=4951,5038
XS Rating Curve= 0
Exp/Cntr=.3,.1

Type RM Length L Ch R = 1 ,88667.88,636.21,532.43,81.26
XS GIS Cut Line= 2
     3267373.303    13866057.765     3263010.684     13866845.46
#Sta/Elev= 30
 3220.09   25.21 3359.69   26.36 4263.62   25.62 4520.48   24.25 4594.45   19.46
 4650.81   17.97 4680.92   15.72 4721.85   16.13 4732.57   17.45 4812.04   10.86
    4960     6.1    4965      .3    4970    -7.5    5000    -9.2    5024    -4.7
    5038     5.5 5149.44   17.46 5239.04   19.21 5275.76   18.41 5383.73   20.23
 5610.79   21.06 6144.58   18.85 6672.14   19.85 6799.33   18.52 6830.49   16.33
 6899.66   17.94 6951.16   14.62 6998.16   13.57 7098.17   21.83 7653.25   24.72
#Mann= 4 ,-1 , 0
 3220.09    .068       04860.355    .118       0    4960     .04       0
    5038    .118       0
#XS Ineff= 1 ,-1
 6375.04 7200.22   19.96
Permanent Ineff=
       F
Bank Sta=4960,5038
XS Rating Curve= 0
Exp/Cntr=.3,.1

Type RM Length L Ch R = 1 ,88135.45,621.75,1127.21,201.4
XS GIS Cut Line= 6
     3267181.408     13865246.67      3265231.38       13865880.
     3265276.515    13865993.996     3265334.487    13866162.358
     3265394.448    13866330.836     3263040.906    13866766.405
#Sta/Elev= 30
 2737.74   25.52 3033.14    25.6 3451.46   24.97 3497.78   19.29 3543.01   25.11
 3953.98   24.47 4053.53   26.75 4155.79    23.2 4175.72   18.88 4201.84    23.7
  4313.2    24.1 4362.43   24.58 4605.81   23.57 4788.04   10.75 4860.95    15.5
 4910.97    14.3 4935.98     3.6 4945.98    -4.2 5037.01    -7.7 5049.02    -4.4
 5062.02     4.6 5089.03    11.4 5423.67   13.92  5670.2   20.75 6737.24   17.03
 6801.86   18.99 6883.62   13.44  6938.6   12.91 7131.41   21.42 7661.04   24.57
#Mann= 6 ,-1 , 0
 2737.74    .068       0 3033.14    .118       0  4313.2    .068       0
 4362.43    .118       0 4910.97     .04       0 5089.03    .118       0
#XS Ineff= 3 ,-1
 3370.73 4030.41   25.51 4108.02 4364.74   24.58 6408.31 7185.82   19.44
Permanent Ineff=
       F       F       F
Bank Sta=4910.97,5089.03
XS Rating Curve= 0
Exp/Cntr=.3,.1

Type RM Length L Ch R = 1 ,87008.24,195.54,1540.38,343.2
XS GIS Cut Line= 6
     3266902.273     13864502.31     3265258.478     13865246.67
     3265168.802    13865351.893     3264875.399    13865734.461
     3264808.761    13866270.165     3262932.353      13866549.3
#Sta/Elev= 30
 2967.76   26.78 3559.04   24.86 3712.76   20.38 4018.59   24.82 4458.65   20.96
  4910.5    23.1  4925.5    14.6  4960.5     6.4  5000.5     4.5  5005.5     1.7
  5010.5    -5.3  5040.5    -8.7  5075.5    -1.3  5080.5     7.6  5089.5     9.6
 5391.89     9.7  5487.6   14.33 5735.41    3.53 5784.85    8.79 5932.54   15.26
 6033.36   14.78 6069.84   18.05 6200.13   17.45 6284.74   20.44 6587.68   16.98
 6728.03    8.75 6795.34    8.18 6916.67   10.68 7043.92   21.23  7829.6   26.09
#Mann= 4 ,-1 , 0
 2967.76    .068       0 3697.04    .118       0  4910.5     .04       0
  5089.5    .118       0
#XS Ineff= 3 ,-1
 3518.34 4031.78   24.78 4105.13 4897.31   23.29 6284.09 7040.29   20.28
Permanent Ineff=
       F       F       F
#Block Obstruct= 2 , 0
                         7523.23           24.91
Bank Sta=4910.5,5089.5
XS Rating Curve= 0
Exp/Cntr=.3,.1

Type RM Length L Ch R = 1 ,85467.86,74.37,1024.06,790.41
XS GIS Cut Line= 6
     3266840.243    13864114.623     3264547.274    13865432.378
     3264474.358    13865781.336     3264388.617    13865850.744
     3264167.066    13866026.128     3262777.278     13866301.18
#Sta/Elev= 30
 1824.89   26.36 2434.07   25.97 3042.72    20.3 3082.76   14.07 3147.97   20.39
 3398.88   22.76 3530.79   18.96 4047.11    20.9 4206.55   18.01 4297.86    7.43
 4427.72     5.5 4548.13    8.66 4654.43   18.44 4826.04   17.81    4860    12.6
    4936     8.9    4951       3    4969     2.5    4971    -1.1    4988   -10.1
    5013   -15.1    5037   -12.8    5049    -8.3    5057     3.3    5064     5.6
 5167.02     5.6 5370.81   19.68 5862.89   21.54 6061.57   25.84 6635.67   26.94
#Mann= 4 ,-1 , 0
 1824.89    .068       0 2883.26    .118       0 4826.04     .04       0
    5064    .118       0
#XS Ineff= 3 ,-1
 2650.37 3383.86   22.39 3420.54 3941.32   20.99 4163.29 4724.31   18.83
Permanent Ineff=
       F       F       F
Bank Sta=4826.04,5064
XS Rating Curve= 0
Exp/Cntr=.3,.1

Type RM Length L Ch R = 1 ,84443.81,508.69,896.15,522.27
XS GIS Cut Line= 6
     3266778.213    13863959.548     3264828.524    13865203.211
     3264711.518    13865148.932     3264615.091    13865109.973
     3264516.024    13865078.211     3262529.158    13865665.373
#Sta/Elev= 30
 2507.11   27.29 3105.43    25.9 3813.08   19.64 3851.38   15.52 3915.24    19.1
  4123.6   16.14 4159.97   17.92 4245.27   16.46  4291.8   19.45 4637.39   20.93
 4812.57   20.09    4887    17.4    4928     7.4    4948     6.1    4961    -6.6
    5000   -16.1    5030   -10.8    5050     1.7    5052     6.7    5073     9.8
 5358.36   11.47  5455.9    6.68 5552.96   12.49 5613.04   20.01 6019.13   24.25
 6255.62    31.4 6540.01   29.11 6602.22   26.23 6690.78   28.92 7228.51   25.96
#Mann= 4 ,-1 , 0
 2507.11    .068       0 3640.25    .118       0    4887     .04       0
    5073    .118       0
#XS Ineff= 1 ,-1
 3393.64 4640.59   20.99
Permanent Ineff=
       F
Bank Sta=4887,5073
XS Rating Curve= 0
Exp/Cntr=.3,.1

Type RM Length L Ch R = 1 ,83547.66,710.29,652.11,184.53
XS GIS Cut Line= 6
      3266731.69    13863587.368     3264495.191    13864776.128
     3264330.913    13864718.805     3264209.887    13864677.132
     3264042.066    13864619.878     3262637.711    13865231.163
#Sta/Elev= 30
 2228.32   27.46 3191.47   24.34 3768.67   15.12 3873.66   19.92 4011.74   17.25
 4086.09   22.15  4217.5    6.58 4259.51   15.85 4301.23   18.67 4432.98   17.51
 4472.61    7.83 4539.16   16.31 4605.71   19.12    4859    14.8    4936     9.6
    4958     5.3    4975    -4.4    5011   -11.9    5035     -10    5060     1.8
    5064     7.5    5120    13.1 5240.43   18.31 5383.39   18.39 5435.14   23.99
 5607.42   20.89 5664.25   25.19 6031.85   30.67 6266.28   25.78 6772.06   25.44
#Mann= 4 ,-1 , 0
 2228.32    .068       0    3546    .118       0    4859     .04       0
    5120    .118       0
#XS Ineff= 3 ,-1
    5478 5783.62   24.16 3510.34 4073.51   19.27 4107.34 4592.71   17.41
Permanent Ineff=
       F       F       F
Bank Sta=4859,5120
XS Rating Curve= 0
Exp/Cntr=.3,.1

Type RM Length L Ch R = 1 ,82895.54,533.39,587.64,390.71
XS GIS Cut Line= 6
     3266592.123    13862703.441     3264607.163     13863944.04
     3264501.977    13864083.283     3264422.557    13864184.936
     3264338.941    13864291.753     3262823.801    13864967.535
#Sta/Elev= 30
 2418.77   28.79 3391.88      26 3712.93   23.41 3974.28   18.43 4435.21   18.54
  4628.2    15.9 4692.33   12.76 4732.17   13.19 4759.53   11.83  4805.5    16.9
  4875.5    15.7  4935.5    10.9  4943.5      .8  4961.5    -8.4  5001.5   -14.2
  5024.5   -11.6  5044.5    -6.4  5059.5      .8  5064.5     8.5  5084.5     8.6
  5103.5    10.6 5238.45    8.98 5296.59    14.4 5370.37   17.96 5899.91    26.7
 6041.77   30.82 6211.36   28.87 6450.42   31.45 6522.83   25.67  6857.7   25.17
#Mann= 4 ,-1 , 0
 2418.77    .068       0 3350.95    .118       0  4935.5     .04       0
  5103.5    .118       0
#XS Ineff= 1 ,-1
  4564.4 4827.87   16.56
Permanent Ineff=
       F
Bank Sta=4935.5,5103.5
XS Rating Curve= 0
Exp/Cntr=.3,.1

Type RM Length L Ch R = 1 ,82307.9 ,30.04,87.01,105.59
XS GIS Cut Line= 6
     3266306.927    13861972.909     3264128.742    13863649.978
     3263989.533    13863807.517     3263878.659    13863935.063
     3263834.754    13863977.374     3262551.897    13864979.606
#Sta/Elev= 30
 1957.97   26.97  2747.7    27.5 2958.98   26.09 3080.51   22.24 3253.41   21.66
 3298.54   21.63 3349.09   24.52 3398.19   20.17 3569.32   18.43 3614.26      16
 4151.94   11.86 4341.24   12.26 4399.44    9.68 4706.98    6.39  4716.5    13.4
  4766.5    12.8  4799.5     9.1  4915.5     7.1  4931.5     4.9  4946.5   -10.3
  4992.5   -13.5  5008.5    -7.6  5023.5     3.4  5066.5     7.7  5084.5    15.7
 5331.61    22.7 5881.26   24.48 6005.31   28.14 6131.19   24.65 6775.13   24.73
#Mann= 4 ,-1 , 0
 1957.97    .068       0 2198.83    .118       0  4766.5     .04       0
  5084.5    .118       0
#Block Obstruct= 1 ,-1
 3020.98 3356.64    24.1
Bank Sta=4766.5,5084.5
XS Rating Curve= 0
Exp/Cntr=.3,.1

Type RM Length L Ch R = 1 ,82220.89,30.14,30,30.18
XS GIS Cut Line= 6
     3266275.442     13861943.58     3264100.701    13863635.184
     3263920.638    13863772.319     3263822.869    13863851.261
      3263786.97    13863887.279     3262480.016    13864890.379
#Sta/Elev= 30
 1960.48   26.82  2207.3   26.75 2319.06   29.46 2385.06   26.65 2913.46   26.44
 3001.76   20.68 3250.36   19.23 3334.24   26.14 3394.96   18.34 3468.24    17.1
  4435.1   11.07  4931.5     4.9  4946.5   -10.3  4992.5   -13.5  5008.5    -7.6
  5023.5     3.4  5134.5    15.8  5248.9    19.6  5440.5   19.59 5566.54   23.31
 6056.16   23.48 6212.26   22.28 6295.62   17.94 6338.42   22.32    6423   25.05
 6488.18   22.23 6550.04   25.02 6610.34   21.72 6682.98   24.63 6766.04   24.34
#Mann= 4 ,-1 , 0
 1960.48    .068       0  2207.3    .118       0  4931.5     .04       0
  5134.5    .118       0
#XS Ineff= 1 ,-1
 5578.85 6390.63    23.3
Permanent Ineff=
       F
#Block Obstruct= 2 , 0
         3342.66   24.57 6426.57           25.03
Bank Sta=4931.5,5134.5
XS Rating Curve= 0
Exp/Cntr=.5,.3

Type RM Length L Ch R = 1 ,82190.89,54.94,54.76,54.98
XS GIS Cut Line= 6
     3266257.023      13861919.9     3264082.403     13863611.41
     3263902.123    13863748.711     3263802.763    13863828.937
     3263767.127    13863864.692      3262461.75    13864866.581
#Sta/Elev= 30
  1955.8   28.37 2139.88   27.11 2289.62   29.92  2453.7   27.46 3182.78   24.05
 3331.12   27.02 3419.56   21.76 3511.64   20.61 3726.66   22.52  4017.3   18.93
 4145.56   20.35 4703.06   17.23    4737    13.3  4766.5     5.7  4931.5     4.9
  4946.5   -10.3  4992.5   -13.5  5008.5    -7.6  5023.5     3.4    5064     7.7
    5108    20.4 5131.42    23.9 5391.18   25.76 5811.08   23.09 6200.52   25.09
 6289.34   22.35 6411.42   27.06 6476.56   23.89 6526.66    26.2 6761.16    25.8
#Mann= 4 ,-1 , 0
  1955.8    .068       0 2139.88    .118       0 4703.06     .04       0
 5131.42    .118       0
#XS Ineff= 2 , 0
       0    4590      24    5166       0    25.2
Permanent Ineff=
       F       F
#Block Obstruct= 2 , 0
                         6229.83           24.57
Bank Sta=4703.06,5131.42
XS Rating Curve= 0
Exp/Cntr=.5,.3

Type RM Length L Ch R = 3 ,82163.1 ,,,
BEGIN DESCRIPTION:
Southern Pacific RR (Just South of I-10)
Southern Pacific RR
END DESCRIPTION:
Bridge Culvert--1,0,-1,-1, 0
Deck Dist Width WeirC Skew NumUp NumDn MinLoCord MaxHiCord MaxSubmerge Is_Ogee
20.4,12,2.6,0, 12, 12, , , .95, 0, 0,0,,
    3296    4336  4714.7  4743.7  4955.1 4955.11 5020.99    5021  5111.4    5982
    6443    6800
    26.6    25.1   27.17   27.41   27.49   30.49   30.48   27.48   27.45    26.2
    26.6    26.6
       0       0   25.17   25.41   25.49   25.49   25.48   25.48   25.45       0
       0       0
    3296    4336  4714.7  4743.7  4955.1 4955.11 5020.99    5021  5111.4    5982
    6443    6800
    26.6    25.1   27.17   27.41   27.49   30.49   30.48   27.48   27.45    26.2
    26.6    26.6
       0       0   25.17   25.41   25.49   25.49   25.48   25.48   25.45       0
       0       0
Pier Skew, UpSta & Num, DnSta & Num=  ,4717.4, 2 ,4714.7, 2 , 0 , 0 , 0 ,,
       1       1
       0      28
       1       1
       0      28
Pier Skew, UpSta & Num, DnSta & Num=  ,4729, 2 ,4729, 2 , 0 , 0 , 0 ,,
       1       1
       0      28
       1       1
       0      28
Pier Skew, UpSta & Num, DnSta & Num=  ,4742.9, 2 ,4742.9, 2 , 0 , 0 , 0 ,,
       1       1
       0      28
       1       1
       0      28
Pier Skew, UpSta & Num, DnSta & Num=  ,4758.4, 2 ,4758.4, 2 , 0 , 0 , 0 ,,
       1       1
       0      28
       1       1
       0      28
Pier Skew, UpSta & Num, DnSta & Num=  ,4773.6, 2 ,4773.6, 2 , 0 , 0 , 0 ,,
       1       1
       0      28
       1       1
       0      28
Pier Skew, UpSta & Num, DnSta & Num=  ,4788.8, 2 ,4788.8, 2 , 0 , 0 , 0 ,,
       1       1
       0      28
       1       1
       0      28
Pier Skew, UpSta & Num, DnSta & Num=  ,4803.8, 2 ,4803.8, 2 , 0 , 0 , 0 ,,
       1       1
       0      28
       1       1
       0      28
Pier Skew, UpSta & Num, DnSta & Num=  ,4819.8, 2 ,4819.8, 2 , 0 , 0 , 0 ,,
       1       1
       0      28
       1       1
       0      28
Pier Skew, UpSta & Num, DnSta & Num=  ,4834.9, 2 ,4834.9, 2 , 0 , 0 , 0 ,,
       1       1
       0      28
       1       1
       0      28
Pier Skew, UpSta & Num, DnSta & Num=  ,4848.3, 2 ,4848.3, 2 , 0 , 0 , 0 ,,
       1       1
       0      28
       1       1
       0      28
Pier Skew, UpSta & Num, DnSta & Num=  ,4863.9, 2 ,4863.9, 2 , 0 , 0 , 0 ,,
       1       1
       0      28
       1       1
       0      28
Pier Skew, UpSta & Num, DnSta & Num=  ,4878.9, 2 ,4878.9, 2 , 0 , 0 , 0 ,,
       1       1
       0      28
       1       1
       0      28
Pier Skew, UpSta & Num, DnSta & Num=  ,4894.1, 2 ,4894.1, 2 , 0 , 0 , 0 ,,
       1       1
       0      28
       1       1
       0      28
Pier Skew, UpSta & Num, DnSta & Num=  ,4909.2, 2 ,4909.2, 2 , 0 , 0 , 0 ,,
       1       1
       0      28
       1       1
       0      28
Pier Skew, UpSta & Num, DnSta & Num=  ,4925.4, 2 ,4925.4, 2 , 0 , 0 , 0 ,,
       1       1
       0      28
       1       1
       0      28
Pier Skew, UpSta & Num, DnSta & Num=  ,4939, 2 ,4939, 2 , 0 , 0 , 0 ,,
       1       1
       0      28
       1       1
       0      28
Pier Skew, UpSta & Num, DnSta & Num=  ,4951, 2 ,4951, 2 , 0 , 0 , 0 ,,
       1       1
       0      28
       1       1
       0      28
Pier Skew, UpSta & Num, DnSta & Num=  ,4954, 2 ,4954, 2 , 0 , 0 , 0 ,,
       1       1
       0      28
       1       1
       0      28
Pier Skew, UpSta & Num, DnSta & Num=  ,5020, 2 ,5020, 2 , 0 , 0 , 0 ,,
       1       1
       0      28
       1       1
       0      28
Pier Skew, UpSta & Num, DnSta & Num=  ,5024.5, 2 ,5024.5, 2 , 0 , 0 , 0 ,,
       1       1
       0      28
       1       1
       0      28
Pier Skew, UpSta & Num, DnSta & Num=  ,5037, 2 ,5037, 2 , 0 , 0 , 0 ,,
       1       1
       0      28
       1       1
       0      28
Pier Skew, UpSta & Num, DnSta & Num=  ,5052.5, 2 ,5052.5, 2 , 0 , 0 , 0 ,,
       1       1
       0      28
       1       1
       0      28
Pier Skew, UpSta & Num, DnSta & Num=  ,5068.8, 2 ,5068.8, 2 , 0 , 0 , 0 ,,
       1       1
       0      28
       1       1
       0      28
Pier Skew, UpSta & Num, DnSta & Num=  ,5084.4, 2 ,5084.4, 2 , 0 , 0 , 0 ,,
       1       1
       0      28
       1       1
       0      28
Pier Skew, UpSta & Num, DnSta & Num=  ,5098.3, 2 ,5098.3, 2 , 0 , 0 , 0 ,,
       1       1
       0      28
       1       1
       0      28
Pier Skew, UpSta & Num, DnSta & Num=  ,5112.2, 2 ,5112.2, 2 , 0 , 0 , 0 ,,
       1       1
       0      28
       1       1
       0      28
BR Coef=-1 , 1 , 1 ,.9, 0 ,,,.8,0,1.2,0,
WSPro=,,,, 1 ,,,, 0 ,,,, 0 ,,,,-1 ,-1 ,-1 , 0 , 0 , 0 , 0 , 0
BC Design=,, 0 ,, 0 ,,,,,,
BC HTab HWMax=29.92

Type RM Length L Ch R = 1 ,82136.12,120.57,120.04,120.7
XS GIS Cut Line= 6
     3266220.066    13861879.368     3264045.567    13863570.784
      3263865.07     13863708.25      3263764.12     13863789.76
     3263728.745    13863825.253     3262424.947     13864825.93
#Sta/Elev= 30
 1951.12   31.79 2095.27   31.71 2352.14   27.98 2732.53   27.59 2766.58   24.83
  3042.8   27.75 3108.88   24.15 3312.56   26.59 3862.81   22.96 4688.57   22.76
 4689.57   22.78 4709.73   20.38 4753.33    6.48 4768.55    5.47 4843.05    4.25
 4940.24    7.52 4962.35  -10.87 4987.68  -11.91 5028.48    -3.5 5042.46    4.54
 5064.87    6.36 5092.86   19.77 5106.78   24.85 5113.01   24.21 5365.76   26.76
 6276.29   20.84 6400.49   24.28 6453.02   22.63 6495.82   25.53 6756.28   25.68
#Mann= 4 ,-1 , 0
 1951.12    .068       0 2095.27    .118       0 4689.57     .04       0
 5113.01    .118       0
#XS Ineff= 2 , 0
       0    4673   24.15    5137       0    25.2
Permanent Ineff=
       F       F
Bank Sta=4688.57,5113.01
XS Rating Curve= 0
Exp/Cntr=.5,.3

Type RM Length L Ch R = 1 ,82016.09,526.68,836.04,771.71
XS GIS Cut Line= 6
      3266146.39    13861784.648     3263972.373    13863475.689
     3263791.009    13863613.816     3263683.697    13863700.463
     3263649.369    13863734.904     3262351.885    13864730.736
#Sta/Elev= 30
 1963.64   22.56 2262.54   25.42 2632.38   21.76 3157.54   25.03 3542.24   20.43
 3599.14   16.97 3901.28   18.87 3970.02   13.97 4068.58   18.53 4194.44    18.6
 4280.66   16.44 4349.06    9.85  4512.7    10.4  4701.9    4.87 4935.13     5.7
 4950.04     .73 4962.35  -10.87 4987.68  -11.91 5028.48    -3.5 5042.46     4.7
 5246.78   16.42 5403.26   21.35 5491.26   21.19 5570.08   16.62 5752.66    21.6
 5883.52   16.25 5940.26   10.36 6060.28    21.4 6148.66   23.52 6768.02   24.83
#Mann= 4 ,-1 , 0
 1963.64    .068       0 2203.86    .118       0 4935.13     .04       0
 5246.78    .118       0
#XS Ineff= 2 ,-1
 5437.65 6149.14   21.34 3515.22 4196.72   18.43
Permanent Ineff=
       F       F
#Block Obstruct= 2 , 0
         3046.45   25.11
Bank Sta=4935.13,5246.78
XS Rating Curve= 0
Exp/Cntr=.3,.1

Type RM Length L Ch R = 1 ,81180.05,430.83,819.69,716.21
XS GIS Cut Line= 6
     3265770.225    13861369.796     3263656.649    13863057.378
     3263492.568    13863056.131     3263392.629    13863052.641
     3263275.144    13863049.861     3261676.246    13864285.205
#Sta/Elev= 30
 2081.48   27.72 2512.42   27.37  2855.2   25.65 2872.29   24.06 2902.63   25.62
 3268.12   23.49 3602.54   24.38 3945.55   22.23 3978.03   19.87 4065.98   19.32
 4582.44   18.27 4662.15   19.98 4750.14   17.69 4822.01   11.58    4836     8.4
    4950     5.5    4953     -.5    4967    -8.3    5000   -15.3    5017   -16.3
    5034     -10    5047     -.5    5050       7 5155.57    8.39 5259.68     4.9
 5397.93   10.17  5436.7    7.42 5663.84    22.5 5796.23   24.83 7188.27   26.32
#Mann= 4 ,-1 , 0
 2081.48    .068       0 2745.36    .118       0    4950     .04       0
    5050    .118       0
Bank Sta=4950,5050
XS Rating Curve= 0
Exp/Cntr=.3,.1

Type RM Length L Ch R = 1 ,80360.35,1690.72,1105.45,617.58
XS GIS Cut Line= 6
      3265553.12    13861044.138     3263521.638    13862672.426
     3263262.092     13862492.92     3263146.855    13862415.192
     3263057.691    13862354.253     3261412.618    13863587.368
#Sta/Elev= 30
  2010.4   27.37 2260.64   25.87 2664.91   26.62 2830.08   24.92 2867.44   22.54
 2899.45   24.83 3002.58   24.45 3892.48   19.35 4005.16   20.81 4070.05   18.68
 4319.98    17.7 4368.46   20.33 4416.71   18.36 4484.52   19.57 4627.97   25.66
 4684.04   23.35  4831.5     7.2  4930.5     5.4  4934.5     1.2  4949.5    -7.8
  5006.5   -12.1  5025.5    -9.3  5044.5     3.9  5046.5     6.4  5069.5     9.2
 5321.51    7.52 5429.49   12.41 5523.12   20.58 5611.17   24.92 7232.41   26.67
#Mann= 4 ,-1 , 0
  2010.4    .068       0 3002.58    .118       0  4930.5     .04       0
  5069.5    .118       0
Bank Sta=4930.5,5069.5
XS Rating Curve= 0
Exp/Cntr=.3,.1

Type RM Length L Ch R = 1 ,79254.91,527.95,979.86,761.33
XS GIS Cut Line= 6
     3263436.347    13860191.226     3263033.152    13860392.823
     3262510.816    13861781.336      3262450.46    13861877.536
     3262304.299    13862160.678      3261187.76    13863060.113
#Sta/Elev= 30
 2850.94   24.24 3469.72   23.81 3855.13   20.37  3966.6   20.89 4011.11   18.91
 4056.54   19.89 4189.17   19.63 4380.65   17.13  4899.5    16.4  4952.5     5.6
  4977.5     3.4  4994.5    -6.6  5011.5    -9.5  5045.5   -11.7  5062.5    -9.3
  5076.5     1.4  5079.5     5.6  5100.5     8.2  5150.5     8.4 5270.48    5.61
 5406.91   17.95 5472.68   20.12 5653.66   19.49 5741.29   21.52 5774.12   23.39
 5838.02   22.15 5903.35      24  5938.2   23.18 6167.24   25.74 6651.23   26.24
#Mann= 4 ,-1 , 0
 2850.94    .068       0 4181.04    .118       0  4899.5     .04       0
  5100.5    .118       0
Bank Sta=4899.5,5100.5
XS Rating Curve= 0
Exp/Cntr=.3,.1

Type RM Length L Ch R = 1 ,78275.05,373.05,1024.79,1138.28
XS GIS Cut Line= 6
     3262707.494    13860377.316     3261730.522    13861943.573
      3261533.11    13862027.056      3261329.13     13862109.47
     3261218.775    13862145.171      3260815.58    13862284.738
#Sta/Elev= 30
 2829.14   24.41  3463.2   21.03 3497.52   20.57 3503.99    18.9 3534.42   20.39
 3786.94   18.36 3895.73   19.37 3924.87    17.5 4017.55   16.32 4159.27   18.05
 4299.34   15.46 4513.86    14.2 4624.13   16.41    4751    11.2    4801      11
    4843     8.8    4890     8.3    4940     8.3    4952     6.4    4956       1
    4992   -12.9    5012   -13.6    5052    -7.8    5068       1    5073     7.9
    5110    12.7    5160    13.5 5377.88   21.37 5464.95   20.97 5652.11   23.92
#Mann= 5 ,-1 , 0
 2829.14    .068       0 3704.26    .118       0    4890     .04       0
    5110    .118       0 5341.58    .068       0
Bank Sta=4890,5110
XS Rating Curve= 0
Exp/Cntr=.3,.1

Type RM Length L Ch R = 1 ,77250.26,941.08,1215.02,1048.96
XS GIS Cut Line= 6
     3262676.479    13860036.151     3261739.983    13861291.753
     3261577.786    13861209.019     3261429.485    13861136.688
     3261328.524    13861093.836     3259541.676    13861123.744
#Sta/Elev= 30
 3169.18   25.13 3508.69   25.19 3706.17   21.99 4152.31   22.54 4426.56   19.65
 4583.95   17.44 4735.56    9.47  4765.5    15.4  4815.5    14.7  4872.5     7.4
  4917.5     4.5  4920.5      .4  4938.5    -8.6  4956.5   -13.3  4974.5     -14
  4992.5   -13.1  5010.5    -7.9  5037.5     5.6  5082.5      12  5132.5      12
 5233.91    6.27 5537.36   14.73  6235.6   16.74 6383.98   11.26 6463.02    2.98
 6578.64    7.41 6641.25   11.44 6692.52   17.95 6762.94   21.58 6979.42   24.64
#Mann= 6 ,-1 , 0
 3169.18    .068       0 4426.56    .118       0  4815.5     .03       0
  5082.5    .068       0 5912.55    .118       0 6903.21    .068       0
#Block Obstruct= 1 ,-1
  6042.9  6690.5   17.34
Bank Sta=4815.5,5082.5
XS Rating Curve= 0
Exp/Cntr=.3,.1

Type RM Length L Ch R = 1 ,76035.24,627.29,1072.4,382.77
XS GIS Cut Line= 6
     3262769.524    13859757.016     3261432.691    13860281.336
      3261361.53    13860176.326     3261292.111    13860065.232
     3261224.358     13859958.42     3259807.592    13860237.748
#Sta/Elev= 30
 3371.09   24.33  3414.5    25.1 3499.06   22.48 3542.99   24.53 3584.41   22.21
 3716.45   24.75 4242.55   22.43  4338.9   23.26 4395.93   22.58 4434.01   20.35
 4602.72    5.97  4650.3    3.66 4744.41     2.9  4881.5     6.7  4934.5     6.8
  4942.5     5.6  4945.5     1.6    4963    -6.1  4998.5   -16.6    5016   -15.7
  5033.5    -8.9  5051.5     1.6  5054.5     6.9  5065.5       8 5328.03    6.87
  5579.3    15.1 6087.28   17.37 6412.75   21.68 6480.89   23.77 6635.45   24.57
#Mann= 3 ,-1 , 0
 3371.09    .068       0  4934.5     .03       0  5065.5    .118       0
Bank Sta=4934.5,5065.5
XS Rating Curve= 0
Exp/Cntr=.3,.1

Type RM Length L Ch R = 1 ,74962.84,504.82,1463.88,1162.89
XS GIS Cut Line= 6
     3263265.764    13859446.866     3261218.775    13859539.911
     3261092.666    13859593.227      3260980.15     13859631.97
     3260784.565    13859694.986      3259574.98    13859726.001
#Sta/Elev= 30
 2752.83   24.98 3003.64   23.01 3350.37   25.76 3475.86   25.39 3560.18   23.14
  3869.3   22.81 4230.16   15.81 4437.73   17.67 4510.11   15.76  4584.3    9.77
 4637.09    8.04  4768.5    7.12  4878.4    9.04  4884.5     7.3  4940.5     5.3
  4943.5     1.3  4979.5   -16.9  5033.5      -6  5059.5       4  5163.5     5.9
  5198.5     9.6  5248.5     9.9 5298.77    7.68 5357.09      13 5442.85   15.95
 5536.55   16.53 5649.75   14.18  5841.8   19.42 5913.92   23.76 6473.32   25.63
#Mann= 4 ,-1 , 0
 2752.83    .068       0 3459.72    .118       0  4940.5     .04       0
  5059.5    .118       0
Bank Sta=4940.5,5059.5
XS Rating Curve= 0
Exp/Cntr=.3,.1

Type RM Length L Ch R = 1 ,73498.96,570.49,1011.03,215.65
XS GIS Cut Line= 6
     3264134.184    13859198.746     3262151.346    13859236.458
     3261906.306    13858929.659     3261811.279     13858812.31
     3261720.893    13858716.449     3259109.755    13858407.863
#Sta/Elev= 30
 2549.06   24.28 3046.45    24.6 3143.09   22.34 3373.54    25.1 3538.38   23.01
 3652.74    24.8 4029.42   24.18    4140   21.05 4275.02   11.33 4473.15   14.18
 4600.02    9.95  4671.5    10.4  4924.5     6.1  4929.5     1.1  4967.5   -14.5
  4986.5   -16.1  5005.5      -8  5045.5     2.8  5059.5     2.9  5075.5     5.6
 5189.65    7.11 5468.36   15.44 5574.59   15.62 5671.38   18.52 5995.46   18.43
 6318.69   23.24 6916.83   25.34 7164.72   23.81 7695.08   24.81 7836.96   26.36
#Mann= 4 ,-1 , 0
 2549.06    .068       0 4029.42    .118       0  4924.5     .04       0
  5075.5    .118       0
Bank Sta=4924.5,5075.5
XS Rating Curve= 0
Exp/Cntr=.3,.1

Type RM Length L Ch R = 1 ,72487.93,629.33,1262.37,747.13
XS GIS Cut Line= 6
     3265049.127    13858919.611     3262816.047    13858842.073
     3262670.629    13858791.534     3262313.039    13858688.997
     3262149.224    13858640.476      3258892.65    13858082.206
#Sta/Elev= 30
 2424.82    25.3 3291.48   24.05 3551.34      26 3656.68   24.11 3886.89   24.98
 3955.61   22.29    4046   24.55 4589.12   23.97    4814    17.4    4836     6.2
    4882     2.9    4885      .6    4903    -1.9    4921     -18    4974   -11.8
    5027      .6    5030     5.8    5122       5    5323     9.2 5444.94    5.07
 5699.34    5.64 5798.99    7.59 5925.37   17.15 6614.83   23.35 7649.71   25.19
 7891.39    23.8 7908.43   21.85 7997.91   25.48 8390.05   24.12 8660.12   25.82
#Mann= 5 ,-1 , 0
 2424.82    .068       0 2923.64    .118       0    4046    .068       0
 4794.24     .04       0    5027    .118       0
Bank Sta=4814,5030
XS Rating Curve= 0
Exp/Cntr=.3,.1

Type RM Length L Ch R = 1 ,71225.56,913.26,1098.97,893.9
XS GIS Cut Line= 6
     3265080.142    13858314.818     3262151.441     13858208.42
     3262137.481    13858120.114     3262113.518    13857984.211
     3262087.194    13857865.101     3258908.157    13857647.996
#Sta/Elev= 30
 1912.27   23.97 3419.68   22.87 3628.23   18.83  3914.3   18.83 4193.99    13.5
 4469.73    12.5 4618.39    6.82 4679.06    9.35    4881     4.5    4931     5.5
    4938       3    4955   -12.7    5001   -19.6    5017   -18.5    5047    -7.3
    5069     5.6    5119     5.4 5192.29   11.27 5344.14   18.14  5817.4   18.95
 6051.41   23.52 6669.12   23.88 6773.65   25.77 6890.21    23.9 7487.88   24.12
 7538.09    21.3 7597.69   23.96 8013.93    24.1 8057.89   26.12 8378.73   24.15
#Mann= 8 ,-1 , 0
 1912.27    .068       0 2429.59    .118       0    4931     .04       0
    5069    .118       0 5404.16    .068       0 5986.14    .118       0
 6180.13    .068       0 7538.09    .118       0
Bank Sta=4931,5069
XS Rating Curve= 0
Exp/Cntr=.3,.1

Type RM Length L Ch R = 1 ,70126.59,1068.93,1093.31,736.83
XS GIS Cut Line= 6
      3268418.01    13857753.948     3262933.761    13857407.683
     3262860.642    13857312.011     3262779.008    13857214.723
     3262703.524    13857130.295     3258846.127    13856826.098
#Sta/Elev= 30
 -674.66    22.8 -424.69   21.63 -385.79   26.19 -334.51   24.58 -274.39   16.84
 -177.71   20.99   371.9   20.58  436.64   24.49  678.78   21.43 2330.74    23.1
 2423.77   25.88 2450.34   22.93 3812.51   23.76 4240.23   17.44 4434.16   18.43
 4572.92    7.78 4691.67    3.36  4911.5     7.1  4936.5     6.1  4966.5      -4
  4984.5   -14.4  5002.5     -18  5063.5     4.4 5163.87   15.45 5347.07   18.07
 6675.65    22.8 7930.42   22.71 7989.86    19.1 8022.42   22.37 9050.55   23.08
#Mann= 7 ,-1 , 0
 -674.66    .068       0 3215.42    .118       0  4911.5     .04       0
  5063.5    .118       0 6230.24    .068       0 7202.76    .118       0
 8369.78    .068       0
#Block Obstruct= 2 ,-1
 -327.55 -176.15   21.01 7843.52 9050.55   22.24
Bank Sta=4911.5,5063.5
XS Rating Curve= 0
Exp/Cntr=.3,.1

Type RM Length L Ch R = 1 ,69033.28,819.25,927.93,370.28
XS GIS Cut Line= 6
     3268509.799    13856889.012     3262984.774    13856401.128
      3262895.61     13856400.23      3262674.11     13856400.23
     3262536.912    13856407.396     3259249.322    13856236.814
#Sta/Elev= 30
  -748.4   22.85 -522.55   24.18 -487.77   20.67 -431.54   24.49  525.75   21.97
  705.34   14.24  918.19   16.01  988.97   10.78 1059.16   17.25 1131.07   19.69
 2047.54    24.4 3358.79   21.64 3719.32   16.38 3952.85   21.17 4112.97   19.66
 4404.79    4.44 4889.25     6.2 4984.75   -27.9 5005.75     -29 5026.75   -25.8
 5047.75   -14.8 5069.75     2.8 5110.75    15.4 5577.27   16.22 5701.13   20.24
 6184.14   21.92  7702.4   22.05  7732.9   17.93 7766.16   21.77 8538.19   21.37
#Mann= 6 ,-1 , 0
  -748.4    .068       0 3802.03    .118       0 4889.25     .04       0
 5110.75    .118       0 7330.93    .068       0  7702.4    .118       0
#XS Ineff= 2 , 0
         3985.61   19.41
Permanent Ineff=
       F       F
#Block Obstruct= 2 ,-1
  517.48  1398.6   21.38 7622.38 8538.19   21.73
Bank Sta=4889.25,5110.75
XS Rating Curve= 0
Exp/Cntr=.3,.1

Type RM Length L Ch R = 1 ,68105.34,959.5,1158.52,930.78
XS GIS Cut Line= 6
     3267317.787    13855182.868      3264651.42    13855075.641
     3263374.317    13855864.634     3263278.732    13855937.287
     3263088.941    13856093.836     3259652.517    13855818.111
#Sta/Elev= 30
  645.14    22.6 2068.68   19.66 2210.66    16.8 3481.46   21.68 4082.64   21.92
 4315.72   21.15 4557.06   16.94  4664.4    7.96 4796.98    2.16  4906.5     1.9
  4931.5       6  4941.5       4    4959    -9.1  4974.5   -14.5    5021   -12.5
    5052    -8.2  5067.5     1.1  5068.5     4.6 5342.58    5.62  5461.1   13.61
 5560.88   15.79 5811.02    12.7 5993.92   14.98  6364.2   20.46 6948.86   22.26
 7892.06   20.62 8089.86   21.26  8135.8   16.66 8171.28   21.42  8628.4   20.85
#Mann= 8 ,-1 , 0
  645.14    .068       0 3481.46    .118       0 4082.64    .068       0
  4931.5     .03       0  5068.5    .068       0 5993.92    .118       0
 7892.06    .068       0 8171.28    .118       0
#XS Ineff= 1 ,-1
 7481.66 8227.38   22.02
Permanent Ineff=
       F
#Block Obstruct= 2 ,-1
  645.14 2811.74   19.53 4699.15  4931.5       6
Bank Sta=4931.5,5068.5
XS Rating Curve= 0
Exp/Cntr=.3,.1

Type RM Length L Ch R = 1 ,66946.82,351.58,988.11,602.94
XS GIS Cut Line= 6
     3265782.881    13854740.107     3264439.959    13854806.651
     3263062.899    13854817.795     3262970.219    13854936.159
     3262786.858    13855161.545     3259652.517    13855151.289
#Sta/Elev= 30
 2053.02   19.07 2975.76   18.84 3031.26    21.6 3088.64   19.11 3353.78   20.37
 3659.62   22.72  4497.8   22.41 4664.94   19.23    4924     2.5    4963   -16.8
    4981     -16    4999   -22.8    5017   -22.5    5053    -3.9    5076     3.2
 5352.74    9.74  5465.2    9.68 5668.94   13.74 5903.94   13.85 6121.12   10.76
 6808.96    18.8  7702.4   21.64 7777.82   19.14 7899.72   21.81 7982.36   17.96
 8005.52   19.92 8143.32   21.28 8203.96   19.78 8233.96   22.06 8349.98   20.89
#Mann= 6 ,-1 , 0
 2053.02    .068       0 3353.78    .118       0    4924     .04       0
    5076    .068       0 5453.38    .118       0 6901.68    .068       0
#XS Ineff= 2 ,-1
  7853.3 8161.37   20.68 5799.51 6449.88    13.6
Permanent Ineff=
       F       F
Bank Sta=4924,5076
XS Rating Curve= 0
Exp/Cntr=.3,.1

Type RM Length L Ch R = 1 ,65958.72,541.76,997.62,849.19
XS GIS Cut Line= 6
     3264486.777    13854487.597     3262273.284    13854484.466
     3262132.055    13854539.895     3262002.236    13854582.076
     3261870.089    13854624.034     3259497.442    13854608.526
#Sta/Elev= 30
 2566.16   20.08 3050.27   22.72  3465.3   22.13 3491.57   23.39 3989.98   19.04
 4130.93   20.91 4193.66   18.33 4524.41   10.49 4611.97   10.25 4846.82    4.82
 4931.75     5.3 4942.25     3.6 4943.25      .5 4958.25   -14.5 4973.75   -19.9
 5018.75   -15.9 5033.75   -13.3 5049.25    -7.5 5068.25     3.2 5442.07   13.95
 5683.15   15.47 5872.12   19.33 6033.09    18.2 6256.29   20.51  6523.6   19.91
 6688.08   21.56 6738.11   15.48  6774.9   20.64 7429.75   21.78 7579.22   20.71
#Mann= 5 ,-1 , 0
 2566.16    .118       0 2666.42    .148       0 3067.47    .118       0
 4931.75     .04       0 5068.25    .068       0
#XS Ineff= 1 ,-1
 6679.71 7442.54   21.46
Permanent Ineff=
       F
Bank Sta=4931.75,5068.25
XS Rating Curve= 0
Exp/Cntr=.3,.1

Type RM Length L Ch R = 1 ,64961.1 ,1107.82,1068.45,1058.91
XS GIS Cut Line= 6
     3264543.014    13853943.974     3262729.566    13853948.003
     3262652.057    13853913.022     3262493.557    13853842.453
     3262366.329    13853802.136     3259311.352    13853802.136
#Sta/Elev= 30
 3014.19   20.56 3087.27    18.5 3125.84   21.13 3293.77   21.73 3375.58   19.97
 3419.78   21.67 3954.87   18.99  4353.5   19.79 4611.89   17.23 4913.25     5.4
 4921.25     2.8 4943.25   -12.5 4963.25   -18.2 4983.25   -18.6 5023.25   -12.8
 5083.25      .2 5086.75     5.4 5137.25     5.7 5272.98     6.2 5391.02   11.72
 5594.78    8.49 6333.91   19.32 7002.87   20.59 7045.05   18.06 7060.05   14.72
 7109.57   20.82 7202.66   21.99 7370.05   20.13 8200.23   20.76 8274.62    18.6
#Mann= 8 ,-1 , 0
 3014.19    .118       0 3224.61    .148       0 4592.32    .118       0
 4913.25     .04       0 5086.75    .068       0 5137.25    .118       0
 5854.82    .068       0  6854.3    .118       0
#XS Ineff= 1 ,-1
 7001.83 8168.11   20.54
Permanent Ineff=
       F
Bank Sta=4913.25,5086.75
XS Rating Curve= 0
Exp/Cntr=.3,.1

Type RM Length L Ch R = 1 ,63892.65,622.94,1262.78,1130.77
XS GIS Cut Line= 6
     3264074.374    13852837.983     3262781.649    13852843.836
      3262658.35     13852829.22      3262527.47     13852817.05
     3262411.858    13852755.295     3259373.382    13852747.626
#Sta/Elev= 30
 3518.58   20.04 4172.98   20.65 4511.05   19.32 4599.43   16.84 4633.39   18.23
 4817.69   11.37 4934.28    3.94 4955.36   -7.15  4981.1  -16.27 5016.02  -22.49
 5065.72    3.99 5450.08    8.58 5709.75   14.29  6279.8   16.38 6429.79   18.94
 6633.78   17.36 6691.49   19.89 6818.09   19.78 6858.59   13.22 6896.33   19.73
 6954.45   20.25 7020.59      17 7091.33   18.89 7940.28   19.78 8069.54   19.25
 8091.66   16.61 8126.33    17.9 8156.33   15.57 8178.03   19.15 8236.48    19.4
#Mann= 7 ,-1 , 0
 3518.58    .068       0 4934.28     .03       0 5065.72    .068       0
 5405.74    .118       0 5594.46    .148       0 7906.23    .068       0
 8094.95    .148       0
#XS Ineff= 1 ,-1
 6769.23 8237.76   19.38
Permanent Ineff=
       F
Bank Sta=4934.28,5065.72
XS Rating Curve= 0
Exp/Cntr=.3,.1

Type RM Length L Ch R = 1 ,62629.87,756.68,846.47,315.04
XS GIS Cut Line= 6
     3264476.253     13852780.22     3262949.441    13852149.156
      3262919.39     13852062.62       3262958.9     13851892.24
     3262661.063    13851693.521     3259853.816     13851461.06
#Sta/Elev= 30
 3168.88   20.67 4205.32   19.25 4546.04    12.7 4681.16    3.86 4912.55    2.67
 4914.17     .24 4945.33   -4.97 4962.95  -10.89 5004.03  -17.12 5022.71  -15.38
 5054.85    -.91 5055.67    1.97 5087.45    8.36  5184.7   10.34 5319.82   14.31
 5582.86   16.94 5785.08   16.86 5818.98   15.17 5901.08   17.28 6643.92   15.44
 6707.36   17.37 6924.88   15.45 6964.46   17.31 7157.12   17.51 7295.04      17
 7367.88   14.39 7490.02    5.02 7548.66   15.28 7587.02   16.34 8262.38    18.7
#Mann= 4 ,-1 , 0
 3168.88    .068       0 4912.55     .03       0 5087.45    .068       0
  5184.7    .148       0
#XS Ineff= 1 ,-1
 7167.83 7818.18   17.42
Permanent Ineff=
       F
Bank Sta=4912.55,5087.45
XS Rating Curve= 0
Exp/Cntr=.3,.1

Type RM Length L Ch R = 1 ,61783.4 ,519.02,2347.25,814.3
XS GIS Cut Line= 6
     3264295.949    13852320.262     3264066.782    13851830.678
        3263724.     13851672.68     3263474.264    13851565.405
     3261720.174    13851275.473     3259887.288      13851293.7
#Sta/Elev= 30
 4003.86    21.4 4387.92   17.98 4691.04    17.7 4772.94    7.31 4921.28    7.97
 4930.44    2.09 4943.61   -1.44 4953.05   -8.99 4977.31  -16.52 5030.85  -15.42
 5078.72    6.11 5166.48    6.34 5229.84   12.44    5312    9.52 5399.02   13.31
 5568.06   14.68  5939.4   12.83 6225.38   15.95 6341.06   14.53  6421.3   17.19
 6809.92   16.98 6882.02   14.68 7061.84   17.38 7159.24   14.56 7208.04   17.31
 7555.92   17.26 7851.56   14.08 7930.68    4.16 8080.46   17.14 8804.56   18.25
#Mann= 5 ,-1 , 0
 4003.86    .068       0 4387.92    .118       0 4921.28     .03       0
 5078.72    .068       0    5312    .148       0
#XS Ineff= 2 ,-1
 7397.44 8784.38   17.42 5723.72 6182.15   15.09
Permanent Ineff=
       F       F
Bank Sta=4921.28,5078.72
XS Rating Curve= 0
Exp/Cntr=.3,.1

Type RM Length L Ch R = 1 ,59436.15,51.3,1094.78,1460.53
XS GIS Cut Line= 6
     3264405.324     13852294.22      3264228.24    13851460.887
     3263769.024     13850698.08      3262706.98     13850713.79
     3262448.316    13850625.086     3260155.063    13849820.936
#Sta/Elev= 30
 2119.27   21.29 2725.16   16.19 3380.59   10.51 3591.46   13.44 4042.36   12.14
 4515.99    7.38 4669.33    2.31 4922.93     4.4 4924.87     .88 4937.32   -1.74
 4955.13   -13.4 4984.27  -17.43 5012.38  -17.69 5038.61     -14  5060.8   -1.02
 5076.03     .86 5077.07    3.76 5479.36    3.57 5620.85   10.42 5864.41   17.32
 6451.42   17.47 6663.68   20.01 6781.22   17.52  6966.5   20.64 7007.04   17.16
 7033.96   11.41 7051.44   12.76 7067.34    17.3 7102.74   19.23 7627.36   19.15
#Mann= 5 ,-1 , 0
 2119.27    .068       0 2725.16    .118       0 2835.32    .068       0
 4922.93     .03       0 5077.07    .148       0
#XS Ineff= 1 ,-1
 6923.08 7167.83   18.66
Permanent Ineff=
       F
#Block Obstruct= 1 ,-1
 5077.19 5488.29    3.76
Bank Sta=4922.93,5077.07
XS Rating Curve= 0
Exp/Cntr=.3,.1

Type RM Length L Ch R = 1 ,58341.37,157.1,69.74,205.41
XS GIS Cut Line= 6
      3264449.68    13852264.312     3264290.907     13851508.05
     3263682.972    13850501.092      3263627.34     13850421.22
     3263448.427    13850256.892     3261789.716    13848273.979
#Sta/Elev= 30
 2879.56   20.93 3495.32    15.7  3956.8   14.16 3990.18   11.83 4134.37   10.34
 4197.47   12.49 4381.15   12.68 4612.95   12.39 4793.43    8.17  4833.6    8.15
 4863.62   10.75 4927.11   10.06 4938.37    1.74 4948.78   -1.09 4961.07  -11.72
 4984.39  -18.65 5015.28  -15.46 5032.79  -11.05 5070.14    1.87 5072.89    5.62
  5249.7    4.76 5311.75    10.2 5399.77   14.82 5704.34   18.25 6094.53   19.37
 6474.24   16.81 6925.46   16.86 7018.85   19.74 7212.33   21.38 7754.14   22.01
#Mann= 4 ,-1 , 0
 2879.56    .068       0 4927.11     .03       0 5072.89    .068       0
 6925.46    .118       0
#Block Obstruct= 2 , 0
                         6058.68           18.82
Bank Sta=4927.11,5072.89
XS Rating Curve= 0
Exp/Cntr=.5,.3

Type RM Length L Ch R = 1 ,58271.63,195.55,181.95,268.89
XS GIS Cut Line= 6
     3264526.295    13852248.559      3264418.19    13851574.979
     3263970.325    13850762.187     3263645.637    13850342.604
     3263531.107      13850175.6     3261889.567     13848172.45
#Sta/Elev= 30
 2814.64   19.77 3537.56   14.69 3882.58   14.39  4012.5   11.54 4316.16   12.69
 4740.92    9.51 4894.94      10 4927.11     8.5 4938.37    1.74 4948.78   -1.09
 4961.07  -11.72 4984.39  -18.65 5015.28  -15.46 5032.79  -11.05 5072.89       4
 5211.04    5.69  5290.7   11.07 5384.76   15.15    5435   15.08 5462.52   17.46
 5529.34   15.27 6007.82   17.98  6239.4   17.48 6396.84   13.59 6726.74    11.6
 6816.38   14.87 7055.12   16.13 7266.68   20.61 7509.42   21.71 7747.74    23.9
#Mann= 4 ,-1 , 0
 2814.64    .068       0 4927.11     .03       0 5072.89    .068       0
 7509.42    .118       0
#XS Ineff= 2 , 0
       0    4817    12.6    5210       0      15
Permanent Ineff=
       F       F
Bank Sta=4927.11,5072.89
XS Rating Curve= 0
Exp/Cntr=.5,.3
